--- Case.prj (project) ---

Proj Title=A2A-010_dx6.25
Current Plan=p01
Default Exp/Contr=0.3,0.1
SI Units
Geom File=g01
Unsteady File=u01
Unsteady File=u02
Plan File=p01
Plan File=p02
Y Axis Title=Elevation
X Axis Title(PF)=Main Channel Distance
X Axis Title(XS)=Station
BEGIN DESCRIPTION:
A2A-010_dx6.25
END DESCRIPTION:
DSS File=dss

--- Case.p01 (plan) ---

Plan Title=Still water (restart)
Program Version=6.60
Short Identifier=init
Simulation Date=01JAN2000,0000,01JAN2000,0001
Geom File=g01
Flow File=u01
Subcritical Flow
K Sum by GR= 0
Std Step Tol= 0.01
Critical Tol= 0.01
Num of Std Step Trials= 20
Max Error Tol= 0.3
Flow Tol Ratio= 0.001
Split Flow NTrial= 30
Split Flow Tol= 0.02
Split Flow Ratio= 0.02
Log Output Level= 0
Friction Slope Method= 1
Unsteady Friction Slope Method= 2
Unsteady Bridges Friction Slope Method= 1
Parabolic Critical Depth
Global Vel Dist= 0 , 0 , 0
Global Log Level= 0
CheckData=True
Encroach Param=-1 ,0,0, 0
Computation Interval=1SEC
Output Interval=1MIN
Instantaneous Interval=1HOUR
Mapping Interval=1MIN
Computation Time Step Use Courant=        -1
Computation Time Step Use Time Series=    0
Computation Time Step Max Courant=1
Computation Time Step Min Courant=0.45
Computation Time Step Count To Double=4
Computation Time Step Max Doubling=3
Computation Time Step Max Halving=6
Computation Time Step Residence Courant=0
Run HTab=-1
Run UNet=-1
Run Sediment= 0
Run PostProcess= 0
Run WQNet= 0
Run RASMapper= 0
UNET Theta= 1
UNET Theta Warmup= 1
UNET ZTol= 0.02
UNET ZSATol= 0.02
UNET MxIter= 20
UNET Max Iter WO Improvement= 0
UNET MaxInSteps= 0
UNET DtIC= 0
UNET DtMin= 0
UNET MaxCRTS= 20
UNET WFStab= 2
UNET SFStab= 1
UNET WFX= 1
UNET SFX= 1
UNET Gravity=9.81
UNET 1D Methodology=Finite Difference
UNET DSS MLevel= 4
UNET Pardiso=0
UNET DZMax Abort= 100
UNET Use Existing IB Tables=-1
UNET Froude Reduction=False
UNET Froude Limit= 1
UNET Froude Power= 10
UNET D1 Cores= 0
UNET D2 Coriolis=0
UNET D2 Theta= 1
UNET D2 Theta Warmup= 1
UNET D2 Z Tol= 0.01
UNET D2 Volume Tol= 0.01
UNET D2 Max Iterations= 20
UNET D2 Equation= 2
UNET D2 RampUpFraction=0.1
UNET D2 TimeSlices= 1
UNET D2 Turbulence Formulation=None
UNET D2 BCVolumeCheck=0
UNET D2 Cores=0
UNET D2 SolverType=Pardiso (Direct)
UNET D2 Name=Strip
UNET D2 Coriolis=0
UNET D2 Theta= 1
UNET D2 Theta Warmup= 1
UNET D2 Z Tol= 0.01
UNET D2 Volume Tol= 0.01
UNET D2 Max Iterations= 20
UNET D2 Equation= 2
UNET D2 RampUpFraction=0.1
UNET D2 TimeSlices= 1
UNET D2 Turbulence Formulation=None
UNET D2 BCVolumeCheck=0
UNET D2 Cores=0
UNET D2 SolverType=Pardiso (Direct)
UNET D1D2 MaxIter= 0
UNET D1D2 ZTol=0.02
UNET D1D2 QTol=1
DSS File=dss
Write IC File=-1
Write IC File at Fixed DateTime=0
Write IC File at Sim End=-1
Echo Input=False
Echo Parameters=False
Echo Output=False
Write Detailed= 1
HDF Write Warmup=0
HDF Write Time Slices=0
HDF Flush=0
HDF Additional Output Variable=Cell Velocity
HDF Additional Output Variable=Face Flow
HDF Compression= 1
HDF Chunk Size= 1
HDF Spatial Parts= 1
HDF Use Max Rows=0
HDF Fixed Rows= 1

--- Case.p02 (plan) ---

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Plan Title=Main
Short Identifier=main
Simulation Date=01JAN2000,0001,01JAN2000,0101
Geom File=g01
Flow File=u02
Write IC File= 0
Write IC File at Sim End=0
Write Detailed= 0

--- Case.u01 (unsteady flow) ---

Flow Title=still water
Program Version=6.60
Use Restart= 0
Initial Storage Elev=Strip           ,1.05746
Boundary Location=                ,                ,        ,        ,                ,Strip           ,                ,Inflow
Interval=1HOUR
Flow Hydrograph= 3
  0.0000  0.0000  0.0000
Stage Hydrograph TW Check=0
Flow Hydrograph Slope= 9.46247e-05
Use DSS=False
Use Fixed Start Time=False
Is Critical Boundary=False
Boundary Location=                ,                ,        ,        ,                ,Strip           ,                ,Outflow
Interval=1HOUR
Stage Hydrograph= 3
  1.0575  1.0575  1.0575
Stage Hydrograph TW Check=0
Use DSS=False
Use Fixed Start Time=False
Is Critical Boundary=False
Precipitation Mode=Disable
Wind Mode=No Wind Forces
Met BC=Precipitation|Mode=None
Met BC=Evapotranspiration|Mode=None

--- Case.u02 (unsteady flow) ---

Flow Title=main
Program Version=6.60
Use Restart=-1
Restart Filename=Case.p01.01JAN2000 0001.rst
Boundary Location=                ,                ,        ,        ,                ,Strip           ,                ,Inflow
Interval=1HOUR
Flow Hydrograph= 3
 20.0000 20.0000 20.0000
Stage Hydrograph TW Check=0
Flow Hydrograph Slope= 9.46247e-05
Use DSS=False
Use Fixed Start Time=False
Is Critical Boundary=False
Boundary Location=                ,                ,        ,        ,                ,Strip           ,                ,Outflow
Interval=1HOUR
Stage Hydrograph= 3
  0.7483  0.7483  0.7483
Stage Hydrograph TW Check=0
Use DSS=False
Use Fixed Start Time=False
Is Critical Boundary=False
Precipitation Mode=Disable
Wind Mode=No Wind Forces
Met BC=Precipitation|Mode=None
Met BC=Evapotranspiration|Mode=None

--- Case.g01 (geometry) ---

Geom Title=A2A-010_dx6.25
Program Version=6.60

Storage Area=Strip           ,500500.0,4000050.0
Storage Area Surface Line= 5
   500000.000000  4000100.000000
   501000.000000  4000100.000000
   501000.000000  4000000.000000
   500000.000000  4000000.000000
   500000.000000  4000100.000000
Storage Area Type= 0
Storage Area Is2D=-1
Storage Area Point Generation Data=,,6.25,6.25
Storage Area 2D Points= 2560
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Storage Area Mannings=0.03
2D Cell Volume Filter Tolerance=0.003
2D Cell Minimum Area Fraction=0.01
2D Face Profile Filter Tolerance=0.003
2D Face Area Elevation Profile Filter Tolerance=0.003
2D Face Area Elevation Conveyance Ratio=0.02
2D Face Area Laminar Depth=0.2

BC Line Name=Inflow
BC Line Storage Area=Strip
BC Line Start Position= 499999.9375 , 4000000.0
BC Line Middle Position= 499999.9375 , 4000050.0
BC Line End Position= 499999.9375 , 4000100.0
BC Line Arc= 2
   499999.937500  4000000.000000   499999.937500  4000100.000000

BC Line Name=Outflow
BC Line Storage Area=Strip
BC Line Start Position= 501000.0625 , 4000000.0
BC Line Middle Position= 501000.0625 , 4000050.0
BC Line End Position= 501000.0625 , 4000100.0
BC Line Arc= 2
   501000.062500  4000000.000000   501000.062500  4000100.000000
LCMann Table=0

Chan Stop Cuts=-1
